--- Muncie2D.prj (project) ---

Proj Title=Muncie2D
Current Plan=p01
Default Exp/Contr=0.3,0.1
English Units
Geom File=g01
Unsteady File=u01
Plan File=p01
Background Map Layer=TerrainWithChannel
Y Axis Title=Elevation
X Axis Title(PF)=Main Channel Distance
X Axis Title(XS)=Station
BEGIN DESCRIPTION:
END DESCRIPTION:
DSS File=dss
DSS Export Rating Curves= 0
DSS Export Rating Curve Sorted= 0
DSS Export Volume Flow Curves= 0
DXF OffsetX= 0
DXF OffsetY= 0
DXF ScaleX= 1
DXF ScaleY= 10

--- Muncie2D.p01 (plan) ---

Plan Title=Peak_flow_plan
Program Version=5.07
Short Identifier=Peak flow
Simulation Date=,0,,6
Geom File=g01
Flow File=u01
Subcritical Flow
K Sum by GR= 0
Std Step Tol= 0.01
Critical Tol= 0.01
Num of Std Step Trials= 20
Max Error Tol= 0.3
Flow Tol Ratio= 0.001
Split Flow NTrial= 30
Split Flow Tol= 0.02
Split Flow Ratio= 0.02
Log Output Level= 0
Friction Slope Method= 1
Unsteady Friction Slope Method= 2
Unsteady Bridges Friction Slope Method= 1
Parabolic Critical Depth
Global Vel Dist= 0 , 0 , 0
Global Log Level= 0
CheckData=True
Encroach Param=-1 ,0,0, 0
Computation Interval=10SEC
Output Interval=1HOUR
Instantaneous Interval=1HOUR
Mapping Interval=15MIN
Computation Time Step Use Courant=        0
Computation Time Step Use Time Series=    0
Computation Time Step Count To Double=0
Computation Time Step Max Doubling=0
Computation Time Step Max Halving=0
Computation Time Step Residence Courant=0
Run HTab=-1
Run UNet=-1
Run Sediment= 0
Run PostProcess=-1
Run WQNet= 0
Run RASMapper= 0
UNET Theta= 1
UNET Theta Warmup= 1
UNET ZTol= 0.02
UNET ZSATol= 0.02
UNET MxIter= 20
UNET Max Iter WO Improvement= 0
UNET MaxInSteps= 0
UNET DtIC= 0
UNET DtMin= 0
UNET MaxCRTS= 20
UNET WFStab= 2
UNET SFStab= 1
UNET WFX= 1
UNET SFX= 1
UNET 1D Methodology=Finite Difference
UNET DSS MLevel= 4
UNET Pardiso=0
UNET DZMax Abort= 100
UNET Use Existing IB Tables=-1
UNET Froude Reduction=False
UNET Froude Limit= 0.8
UNET Froude Power= 4
UNET D1 Cores= 0
UNET D2 Coriolis=0
UNET D2 Cores= 0
UNET D2 Theta= 1
UNET D2 Theta Warmup= 1
UNET D2 Z Tol= 0.01
UNET D2 Volume Tol= 0.01
UNET D2 Max Iterations= 20
UNET D2 Equation= 1
UNET D2 RampUpFraction=0.1
UNET D2 TimeSlices= 1
UNET D2 BCVolumeCheck=0
UNET D2 Name=Muncie_Geom
UNET D2 Theta= 1
UNET D2 Theta Warmup= 1
UNET D2 Z Tol= 0.01
UNET D2 Volume Tol= 0.01
UNET D2 Max Iterations= 20
UNET D2 Equation= 1
UNET D2 RampUpFraction=0.1
UNET D2 TimeSlices= 1
UNET D2 BCVolumeCheck=0
UNET D1D2 MaxIter= 0
UNET D1D2 ZTol=0.01
UNET D1D2 QTol=0.1
UNET D1D2 MinQTol=1
DSS File=dss
Write IC File= 0
Write IC File at Fixed DateTime=0
Write IC File at Sim End=0
Echo Input=False
Echo Parameters=False
Echo Output=False
Write Detailed= 0
Computation Level Output Depth=True
HDF Write Warmup=0
HDF Write Time Slices=0
HDF Flush=0
HDF Face Node Velocities=-1
HDF Compression= 1
HDF Chunk Size= 1
HDF Spatial Parts= 1
HDF Use Max Rows=0
HDF Fixed Rows= 1
Calibration Method= 0
Calibration Iterations= 20
Calibration Max Change=0.05
Calibration Tolerance=0.2
Calibration Maximum=1.5
Calibration Minimum=0.5
Calibration Optimization Method= 1
WQ AD Non Conservative
WQ ULTIMATE=-1
WQ Max Comp Step=1HOUR
WQ Output Interval=15MIN
WQ Output Selected Increments= 0
WQ Output face flow=0
WQ Output face velocity=0
WQ Output face area=0
WQ Output face dispersion=0
WQ Output cell volume=0
WQ Output cell surface area=0
WQ Output cell continuity=0
WQ Output cumulative cell continuity=0
WQ Output face conc=0
WQ Output face dconc_dx=0
WQ Output face courant=0
WQ Output face peclet=0
WQ Output face adv mass=0
WQ Output face disp mass=0
WQ Output cell mass=0
WQ Output cell source sink temp=0
WQ Output nsm pathways=0
WQ Output nsm derived pathways=0
WQ Output MaxMinRange=-1
WQ Daily Max Min Mean=-1
WQ Daily Range=0
WQ Daily Time=0
WQ Create Restart=0
WQ Fixed Restart=0
WQ System Summary=0
WQ Write To DSS=0
WQ Use Fixed Temperature=0
Sorting and Armoring Iterations= 10
XS Update Threshold= 0.02
Bed Roughness Predictor= 0
Hydraulics Update Threshold= 0.02
Energy Slope Method= 1
Volume Change Method= 1
Sediment Retention Method= 0
XS Weighting Method= 0
Number of US Weighted Cross Sections= 1
Number of DS Weighted Cross Sections= 1
Upstream XS Weight=0
Main XS Weight=1
Downstream XS Weight=0
Number of DS XS's Weighted with US Boundary= 1
Upstream Boundary Weight= 1
Weight of XSs Associated with US Boundary= 0
Number of US XS's Weighted with DS Boundary= 1
Downstream Boundary Weight= 0.5
Weight of XSs Associated with DS Boundary= 0.5
Percentile Method= 0
Sediment Output Level= 3
Mass or Volume Output= 0
Output Increment Type= 1
Profile and TS Output Increment= 1
XS Output Flag= 0
XS Output Increment= 10
Write Gradation File= 0
Read Gradation Hotstart= 0
Write HDF5 File= 1
Write Binary Output= 1
Write DSS Sediment File= 0
SV Curve= 0
Specific Gage Flag= 0

--- Muncie2D.u01 (unsteady flow) ---

Flow Title=Muncie_Peak_Flow
Program Version=5.07
Use Restart= 0
Boundary Location=                ,                ,        ,        ,                ,Muncie_Geom     ,                ,outlet
Interval=1HOUR
Stage Hydrograph= 7
     930     930     930     930     930     930     930
Stage Hydrograph Use Initial Stage=-1
Stage Hydrograph TW Check=0
Use DSS=False
Use Fixed Start Time=False
Is Critical Boundary=False
Boundary Location=                ,                ,        ,        ,                ,Muncie_Geom     ,                ,inlet
Interval=1HOUR
Flow Hydrograph= 7
   20000   20000   20000   20000   20000   20000   20000
Stage Hydrograph TW Check=0
Flow Hydrograph Slope= 0.0001
Use DSS=False
Use Fixed Start Time=False
Is Critical Boundary=False

--- Muncie2D.g01 (geometry) ---

Geom Title=Muncie_base2D
Program Version=5.07

Storage Area=Muncie_Geom     ,409230.4562239,1803255.155042
Storage Area Surface Line= 6
414421.7351049921800819.12925698
405441.887976495 1800724.6379195
403127.9134985191804933.83669128
407833.6931832581805557.81395557
408577.1206412481807466.91484153
414421.7351049921800819.12925698
Storage Area Type= 1
Storage Area Is2D=-1
Storage Area Point Generation Data=0,0,50,50
Storage Area 2D Points= 19407
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Storage Area Mannings=0.03
2D Cell Volume Filter Tolerance=0.01
2D Cell Minimum Area Fraction=0.01
2D Face Profile Filter Tolerance=0.01
2D Face Area Elevation Profile Filter Tolerance=0.01
2D Face Area Elevation Conveyance Ratio=0.02
2D Face Area Laminar Depth=0.2

BreakLine Name=breakline_1
BreakLine Near Repeats=1
BreakLine Protection Radius=0
BreakLine Polyline= 4
409010.6110160081801949.94013548409051.3970494861802463.84415732
409858.9605123641802390.42929705410160.777160106 1801737.8527614

BreakLine Name=breakline_2
BreakLine Near Repeats=1
BreakLine Protection Radius=0
BreakLine Polyline= 3
 408814.838055311802390.42929705408635.3795080041802651.45991132
408994.2966026161802830.91845862

BreakLine Name=breakline_leftba
BreakLine Near Repeats=1
BreakLine Protection Radius=0
BreakLine Polyline= 6
414590.1403958881800212.45510929411302.7860975081803295.87924028
 406465.562526941805049.67867986404964.6364949251804715.23320534
405690.6278908451802618.83108453404581.2477802261801558.39421409

BreakLine Name=breakline_rightb
BreakLine Near Repeats=1
BreakLine Protection Radius=0
BreakLine Polyline= 6
414549.3543624091800432.69969008413146.3148107431800440.85689677
411449.6158180311803459.02337419409393.9997307071802994.06259254
405823.0141188671805288.38820868404499.6757132691801705.22393461

BreakLine Name=tribu_bankright
BreakLine Near Repeats=1
BreakLine Protection Radius=0
BreakLine Polyline= 6
408281.0147425541804202.54323851408311.9051225981804590.87944478
408439.8795542091805120.42881697408885.5836091311805901.51414094
409017.9709521781806431.06351312408987.0805721331806603.16705908

BreakLine Name=road1
BreakLine Near Repeats=1
BreakLine Protection Radius=0
BreakLine Polyline= 6
 412574.775633051801447.79206206412442.2245197431801329.44285375
 412368.848010591801225.29555044412295.4715014381801182.68983545
412226.8289606181801097.47840546412068.2410214831801009.89999131

BreakLine Name=road2
BreakLine Near Repeats=1
BreakLine Protection Radius=0
BreakLine Polyline= 6
 412761.76738218 1801585.0771437412967.6950046391801724.72920951
413306.1737404061801433.59015706413585.4778720181801459.62698289
413495.5324737021801660.82063702413505.0004103671801916.45492697

BreakLine Name=ridge1
BreakLine Near Repeats=1
BreakLine Protection Radius=0
BreakLine Polyline= 6
412342.4186535251802802.81653305411788.4283347081802851.69803177
411793.8596123431802927.73591866412434.7503733281803058.08658191
 411989.385607221803177.57468989411826.4472781561803378.53196241

BC Line Name=outlet
BC Line Storage Area=Muncie_Geom
BC Line Start Position= 402980.381796636 , 1803620.06744422
BC Line Middle Position= 404203.59836005 , 1802180.19319808
BC Line End Position= 405426.814923465 , 1800740.31895193
BC Line Arc= 2
402980.3817966361803620.06744422405426.8149234651800740.31895193

BC Line Name=inlet
BC Line Storage Area=Muncie_Geom
BC Line Start Position= 414544.984060369 , 1800146.73922907
BC Line Middle Position= 414498.737375412 , 1800406.04137754
BC Line End Position= 414452.490690456 , 1800665.34352602
BC Line Arc= 2
414544.9840603691800146.73922907414452.4906904561800665.34352602
LCMann Table=0

LCMann Region Name=0
LCMann Region Table=0
LCMann Region Polygon= 6
         412732.        1804610.         414469.        1802943.
         414593.        1800411.         411802.        1802161.
         411504.        1803429.         412732.        1804610.

LCMann Region Name=1
LCMann Region Table=0
LCMann Region Polygon= 6
         409385.        1802639.         411277.        1803301.
         414603.        1800217.         414874.        1798892.
         409473.        1801121.         409385.        1802639.

LCMann Region Name=2
LCMann Region Table=0
LCMann Region Polygon= 6
         408161.        1804209.         409436.        1807302.
         412732.        1804610.         411504.        1803429.
         409810.        1802894.         408161.        1804209.

LCMann Region Name=3
LCMann Region Table=0
LCMann Region Polygon= 6
         404578.        1801617.         405680.        1802516.
         404957.        1804702.         406451.        1805075.
         409473.        1801121.         404578.        1801617.

LCMann Region Name=4
LCMann Region Table=0
LCMann Region Polygon= 6
         404489.        1801758.         404735.        1804709.
         406377.        1805222.         414603.        1800217.
         406451.        1805075.         404489.        1801758.

LCMann Region Name=5
LCMann Region Table=0
LCMann Region Polygon= 6
402883.905406507 1803654.7192238         404793.        1807035.
         409436.        1807302.         404897.        1804951.
         404689.        1801833.402883.905406507 1803654.7192238

Chan Stop Cuts=-1
Use User Specified Reach Order=0
Composite Channel Slope=5
